--- BrshCrk.prj (project) ---

Proj Title=BrshCrk
Current Plan=p01
Default Exp/Contr=0,0
English Units
Geom File=g01
Flow File=f01
Plan File=p01
BEGIN DESCRIPTION:
END DESCRIPTION:
DSS Export Rating Curves= 0
DSS Export Rating Curve Sorted= 0
DSS Export Volume Flow Curves= 0
DXF OffsetX= 0
DXF OffsetY= 0
DXF ScaleX= 0
DXF ScaleY= 0

--- BrshCrk.p01 (plan) ---

Plan Title=Floodplain
Program Version=4.00
Geom File=g01
Flow File=f01
K Sum by GR=0
Std Step Tol=0.01
Critical Tol=0.01
Num of Std Step Trials=20
Max Error Tol=0.3
Flow Tol Ratio=0.001
Split Flow NTrial=30
Split Flow Tol=0.02
Split Flow Ratio=0.02
Log Output Level=0
Friction Slope Method=1
Unsteady Friction Slope Method=2
Unsteady Bridges Friction Slope Method=1
Global Log Level=0
CheckData=False
Run HTab=0
Run UNet=0
Run PostProcess=0
UNET Theta=0
UNET Theta Warmup=0
UNET ZTol=0
UNET ZSATol=0
UNET MxIter=0
UNET MaxInSteps=0
UNET DtIC=0
UNET DtMin=0
UNET MaxCRTS=0
UNET WFStab=0
UNET SFStab=0
UNET WFX=0
UNET SFX=0
UNET DSS MLevel=0
UNET DZMax Abort=0
UNET Convert EG Bridges=0
UNET Use Existing IB Tables=0
UNET Froude Limit=0
UNET Froude Power=0
Write IC File=0
Echo Input=False
Echo Output=False
Write Detailed=0

--- BrshCrk.f01 (steady flow) ---

Flow Title=NFF Regression Equation
Program Version=4.00
Number of Profiles=1
Profile Names=P100yr
River Rch & RM=BrshCrk,Main      ,35022.4
6574.976
River Rch & RM=BrshCrk,Main      ,17002.1
7197.613
River Rch & RM=BrshCrk,Main      ,16281.9
8954.600
River Rch & RM=BrshCrk,Main      ,310.2
9269.585
Boundary for River Rch & Prof#=BrshCrk,Main      ,1
Up Type=0
Dn Type=3
Dn Slope=0.025631

--- BrshCrk.g01 (geometry) ---

Geom Title=USGS 3m DEM
Program Version=4.10

River Reach=BrshCrk         ,Main
Reach XY= 30
      1949673.85      155988.697     1950390.468      157664.393
      1950079.27      158866.216     1950448.911      158825.335
     1950888.619      158098.726     1951866.827      157753.953
     1952125.172      158091.925     1951978.436      159061.942
     1952472.212      159512.308     1953470.197      158797.334
     1954645.676      158660.487      1955415.34       159210.26
     1955631.353      161090.175     1955382.832      161575.299
     1956510.259      162832.362      1957141.63      164699.508
     1956983.764      165009.764     1956257.366      164818.116
     1956127.481      165138.318     1954847.213       165543.34
     1952739.498      167321.492     1951669.066      167378.216
     1951138.583      167002.408     1950637.147      168135.251
     1949755.051      168471.685     1949755.454      169212.242
     1950509.862       169353.81     1951579.433       171041.85
     1951343.721      172857.186     1950629.418      173946.419

Type RM Length L Ch R = 1 ,35022.4 ,499.4,499.8,500.1
XS GIS Cut Line= 2
     1949359.169      156150.617     1950135.912      155970.032
#Sta/Elev= 30
       0 2403.05      10 2401.52    39.9 2401.48    49.8 2401.05    59.8 2399.74
    79.8 2396.12   109.6 2386.55   139.6 2374.43   159.5 2371.43   169.5 2368.52
   189.4 2360.88   199.4 2359.02   229.3 2354.55   269.1  2350.8   289.1 2350.17
     319 2348.45   338.9 2348.14   339.2    2344   359.2    2344   368.8  2348.1
   378.8 2348.63   388.8 2350.35   428.6  2360.1   438.6 2364.14   448.6 2367.25
   508.4 2382.37   518.4  2384.7   528.3 2385.87   687.8  2389.8   797.5 2390.92
#Mann= 3 , 0 , 0
       0      .1       0   339.2    .045       0   359.2      .1       0
Bank Sta=339.2,359.2
XS Rating Curve= 0 ,0
Exp/Cntr=0.3,0.1

Type RM Length L Ch R = 1 ,34522.5 ,546.9,532.2,517.7
XS GIS Cut Line= 3
     1949467.924      156621.965     1949875.441      156534.962
     1950273.949      156446.405
#Sta/Elev= 30
       0 2389.72    29.8  2384.3    39.7 2383.92    49.6 2382.43    69.4 2377.64
    79.4 2376.27   148.8 2376.34   218.3 2377.74     248 2377.35     258 2375.44
   317.5 2360.03   327.4 2355.29   367.1 2344.49     377 2342.62   396.9  2341.8
   402.1  2341.8   422.1 2341.98   476.4 2347.22     566 2366.57     576 2369.31
     586  2373.5   615.8 2378.33   655.7 2381.55   675.6  2384.1   685.5 2383.95
   715.4 2380.01   725.4 2379.92   735.3 2380.61   765.2    2385   824.9 2386.46
#Mann= 3 , 0 , 0
       0      .1       0   402.1    .045       0   422.1      .1       0
Bank Sta=402.1,422.1
XS Rating Curve= 0 ,0
Exp/Cntr=0.3,0.1

Type RM Length L Ch R = 1 ,33990.3 ,191.8,188.7,184.1
XS GIS Cut Line= 3
     1949548.533      157286.294     1949738.096      157254.256
     1950279.443      156709.581
#Sta/Elev= 30
       0 2393.72    76.9 2394.71   134.6 2396.84   153.8 2398.18   163.4  2399.6
     272 2409.76     302 2411.67   311.9 2411.22   321.9 2407.67   351.8 2392.19
   371.8 2386.61   391.7 2375.71   421.6 2363.56   451.6  2353.7   481.5 2346.16
   494.2 2344.31   501.4 2342.63   511.4  2341.8   514.2  2341.8   541.3 2341.91
   551.3 2342.56   591.2 2351.16   611.1 2354.23   631.1 2360.15     641 2361.74
     651 2362.39   710.9 2379.38   720.8 2381.68   850.5 2388.62   960.2 2390.78
#Mann= 3 , 0 , 0
       0      .1       0   494.2    .045       0   514.2      .1       0
Bank Sta=494.2,514.2
XS Rating Curve= 0 ,0
Exp/Cntr=0.3,0.1

Type RM Length L Ch R = 1 ,33801.6 ,412.5,430.1,449.2
XS GIS Cut Line= 3
     1949865.681      157456.818     1950118.713      157131.858
     1950351.617      156795.402
#Sta/Elev= 30
       0 2400.39    39.2 2405.12   107.9 2407.61   137.3 2407.46   225.5 2405.01
   235.4 2402.18   245.2 2398.45   274.6 2386.05   284.4 2384.33   294.2  2381.5
     353 2358.28   372.6 2351.26   401.9 2341.93   421.9 2340.64   471.7 2340.49
   491.7 2340.62   501.7 2341.58   511.7 2344.31   521.6 2345.58   531.6 2348.75
   541.6 2353.34   551.6 2360.12   571.5 2369.86   581.5 2374.02   601.5 2380.12
   611.5 2381.96   641.4 2384.71   671.4 2385.38   741.2 2389.52   821.1 2392.66
#Mann= 3 , 0 , 0
       0      .1       0   401.9    .045       0   421.9      .1       0
Bank Sta=401.9,421.9
XS Rating Curve= 0 ,0
Exp/Cntr=0.3,0.1

Type RM Length L Ch R = 1 ,33371.4 ,328.9,340.6,352.4
XS GIS Cut Line= 2
     1949928.088      157545.561     1950736.259      157369.658
#Sta/Elev= 30
       0 2392.06    49.8 2393.84    99.6 2394.98   169.4 2394.87   189.3 2395.26
   239.2 2398.42     269 2401.42     279 2401.57     289 2397.78   358.7 2360.53
   368.7 2350.45   378.7 2344.69   388.6 2339.65   398.6  2336.3   408.7 2335.28
   428.7  2335.2   438.5 2335.19   448.4 2335.87   458.4 2337.38   488.3 2343.34
   518.2 2350.03   538.1 2357.47   587.9 2370.38   607.9  2375.2   617.8 2376.62
   657.7 2380.45   697.6 2384.78   707.5 2386.88   787.2  2396.2   827.1 2398.97
#Mann= 3 , 0 , 0
       0      .1       0   408.7    .045       0   428.7      .1       0
Bank Sta=408.7,428.7
XS Rating Curve= 0 ,0
Exp/Cntr=0.3,0.1

Type RM Length L Ch R = 1 ,33030.8 ,420.1,424.1,428.1
XS GIS Cut Line= 3
     1949946.349        157676.1     1950557.757      157828.285
     1950783.102      157581.241
#Sta/Elev= 30
       0 2379.47    78.8 2375.79   137.8 2376.37   177.2 2374.36   196.9 2374.98
   216.6 2373.62   295.3 2365.74   324.9 2364.05   334.7 2362.73   344.6 2360.45
   393.8  2335.3   403.6 2332.07   408.7 2331.49   413.5 2330.94   428.7  2330.8
     443 2330.78   472.6 2331.92   511.9 2335.84   531.6 2340.12   600.5 2351.86
   610.4 2355.31   689.1 2368.98   718.6 2373.02   738.2 2374.58   767.8 2375.71
   807.1 2378.27   846.4 2382.29   885.8 2385.37   915.3 2388.58   964.4 2391.07
#Mann= 3 , 0 , 0
       0      .1       0   408.7    .045       0   428.7      .1       0
Bank Sta=408.7,428.7
XS Rating Curve= 0 ,0
Exp/Cntr=0.3,0.1

Type RM Length L Ch R = 1 ,32606.5 ,821.9,790,758.2
XS GIS Cut Line= 2
     1949960.922      158028.547     1950485.669      158252.799
#Sta/Elev= 30
       0 2385.27    49.2 2379.27      59 2377.62    68.9 2375.22    78.7 2372.26
    88.6 2368.06    98.4 2362.39   108.2 2359.13   118.1 2356.46   127.9 2354.03
   137.7 2351.87   177.1 2343.42   186.9 2341.82   226.3 2338.05     246 2336.35
   265.6 2334.38   275.5 2333.62   344.4 2330.52   354.2 2329.66     364 2329.13
   383.7 2328.41   403.1  2327.5   423.1  2327.4   442.8 2327.39   452.6 2329.05
   521.5 2347.37   531.3 2350.13   541.1 2354.45     551  2355.5   570.7 2355.42
#Mann= 3 , 0 , 0
       0      .1       0   403.1    .045       0   423.1      .1       0
Bank Sta=403.1,423.1
XS Rating Curve= 0 ,0
Exp/Cntr=0.3,0.1

Type RM Length L Ch R = 1 ,31816.5 ,587.6,555.4,523.2
XS GIS Cut Line= 4
     1949601.873      158852.009     1949864.241      158963.482
     1950319.194      158487.545     1950365.622      158443.438
#Sta/Elev= 30
       0  2354.7    29.5  2354.7    39.3 2355.39    78.6 2367.88    88.5 2369.49
    98.3 2370.02   167.1 2369.51   235.9  2366.6   285.1 2368.18     315 2366.73
   354.9 2364.08   364.9 2362.87   374.8 2360.41   414.8    2348   434.7 2340.23
   444.7  2337.2   454.7 2335.98   474.6 2330.16   484.6 2327.94   490.9 2327.61
   504.5 2327.37   510.9 2327.38   534.5 2327.45   654.2 2330.76     704  2334.6
     724 2335.24   773.9 2340.32   863.7 2345.04   961.8 2351.38  1007.5 2353.27
#Mann= 3 , 0 , 0
       0      .1       0   490.9    .045       0   510.9      .1       0
Bank Sta=490.9,510.9
XS Rating Curve= 0 ,0
Exp/Cntr=0.3,0.1

Type RM Length L Ch R = 1 ,31260.9 ,336.8,321.7,306.5
XS GIS Cut Line= 3
       1951004.4      159626.277     1950651.955      159040.917
     1950356.337      158524.688
#Sta/Elev= 30
       0 2368.06    19.8 2365.14    49.5 2365.62   108.9 2360.61   158.4 2360.22
     198 2361.86   227.8 2366.16   237.7 2365.67   257.5 2366.66   316.9 2376.45
   346.6 2379.49   356.5  2378.4     406 2381.32     505 2377.46   554.5 2377.44
   722.9 2361.58   752.7 2357.55     832 2352.01   861.7 2347.03   891.5 2340.53
   901.4 2339.46   982.3 2320.51  1002.3 2316.25  1050.1 2314.99    1070 2316.75
  1089.8 2324.25  1109.6 2329.82  1129.4 2332.67    1179 2344.61  1278.2 2349.49
#Mann= 3 , 0 , 0
       0      .1       0   982.3    .045       0  1002.3      .1       0
Bank Sta=982.3,1002.3
XS Rating Curve= 0 ,0
Exp/Cntr=0.3,0.1

Type RM Length L Ch R = 1 ,30939.3 ,276.9,279.3,281.8
XS GIS Cut Line= 2
     1951164.193      158752.187     1950484.015      158417.902
#Sta/Elev= 30
       0 2396.25    19.9 2395.37    49.9 2392.72    59.8 2391.03   109.7 2385.34
   139.6 2382.75   189.5 2377.19   209.4 2376.07   239.3 2372.03   329.1 2365.63
     359 2361.99     369 2360.27   378.9 2357.07   388.9 2352.75   418.8 2337.82
   428.8 2329.53   438.8 2325.97   478.7  2317.5   518.8 2312.54   528.5 2312.41
   538.8 2312.43   558.4 2312.94   568.4 2314.43   588.4 2318.79   598.3 2321.52
   608.3 2326.09   638.2 2334.52     698 2349.82     708 2351.19   757.9 2352.63
#Mann= 3 , 0 , 0
       0      .1       0   518.8    .045       0   538.8      .1       0
Bank Sta=518.8,538.8
XS Rating Curve= 0 ,0
Exp/Cntr=0.3,0.1

Type RM Length L Ch R = 1 ,30659.8 ,522.2,549.1,575.9
XS GIS Cut Line= 3
     1951147.943      158482.902     1950593.122      158139.331
     1950637.229       157812.01
#Sta/Elev= 30
       0 2384.76    39.6 2381.56      89 2374.68   158.2 2370.68     178 2364.81
   197.8 2356.55   217.5 2351.64   237.3 2345.14   296.6 2335.24   336.2 2322.41
   365.8 2315.55   385.6    2310   424.3  2308.9   444.3 2309.42   474.6 2314.26
   484.5 2316.87   504.3 2323.83   514.2 2328.46     524 2337.16   533.9 2344.35
   553.7 2354.38   563.6  2356.8   652.6 2359.58   710.9 2360.14   749.7 2362.55
   778.9  2363.2   846.9 2359.49   895.4 2363.49   953.7 2365.47   982.9 2368.99
#Mann= 3 , 0 , 0
       0      .1       0   424.3    .045       0   444.3      .1       0
Bank Sta=424.3,444.3
XS Rating Curve= 0 ,0
Exp/Cntr=0.3,0.1

Type RM Length L Ch R = 1 ,30110.6 ,311.1,296.6,282.6
XS GIS Cut Line= 2
     1951216.591      158526.388      1951257.05      157791.117
#Sta/Elev= 30
       0 2392.91    29.8 2390.83    59.7 2384.43    69.7 2383.68   139.3 2363.49
   149.3 2361.12   159.2 2360.49     199 2348.02   228.9 2336.95   248.8 2331.42
   258.7    2331   288.6 2323.44   328.4 2316.16   338.3 2314.72   348.3 2314.58
   388.1 2308.44   409.7 2307.75   429.7 2307.64   437.8  2307.6   457.8 2307.72
   467.7 2309.44   497.6 2320.18   527.4 2332.79   537.4 2332.89   577.2 2350.06
   626.9 2370.02   636.9 2370.33   666.7 2379.77   686.6 2381.87   736.4 2380.69
#Mann= 3 , 0 , 0
       0      .1       0   409.7    .045       0   429.7      .1       0
Bank Sta=409.7,429.7
XS Rating Curve= 0 ,0
Exp/Cntr=0.3,0.1

Type RM Length L Ch R = 1 ,29814.1 ,392.5,397.8,402.6
XS GIS Cut Line= 3
     1951425.539      158520.821     1951584.371      158188.081
     1951288.359      157671.597
#Sta/Elev= 30
       0 2404.77    49.8 2400.33    99.6 2397.74   149.5 2388.51   159.4 2387.37
   169.4 2387.91   199.3 2382.56   239.2 2370.75   269.1 2363.34     279 2364.08
   348.8  2348.9   378.6 2344.52     458 2316.04   477.8 2307.51   484.5 2306.32
   504.5 2304.82   507.6  2304.7   547.3 2305.19   577.1 2309.16   626.7 2312.83
   656.4 2317.51   686.2 2325.03     706 2328.38   745.7 2342.76   775.5 2355.05
   805.3 2369.03   815.2 2371.45   844.9 2384.06   864.8    2385     964 2378.11
#Mann= 3 , 0 , 0
       0      .1       0   484.5    .045       0   504.5      .1       0
Bank Sta=484.5,504.5
XS Rating Curve= 0 ,0
Exp/Cntr=0.3,0.1

Type RM Length L Ch R = 1 ,29416.2 ,360.1,392,423.4
XS GIS Cut Line= 3
      1951473.69      158491.862     1951809.549       157925.76
     1951579.728       157208.44
#Sta/Elev= 30
       0 2403.42   169.6  2394.7   189.5 2392.34   249.3 2377.52   289.2  2379.5
   349.1 2376.71     369  2378.8   418.9 2375.29   468.7 2376.23   558.5 2372.88
   588.4 2366.55   598.4 2359.02   618.3 2337.79   628.3 2329.54   658.2 2316.29
   777.2 2299.78   808.1 2298.18   828.1 2297.82   846.5 2297.64   886.2 2301.16
   915.9  2313.1   935.7 2324.85   975.4 2355.26   995.2 2362.87  1024.9 2383.25
  1034.8 2385.51  1223.2 2379.16  1302.4  2383.4  1391.6  2394.3  1411.5 2398.53
#Mann= 3 , 0 , 0
       0      .1       0   808.1    .045       0   828.1      .1       0
Bank Sta=808.1,828.1
XS Rating Curve= 0 ,0
Exp/Cntr=0.3,0.1

Type RM Length L Ch R = 1 ,29024   ,523.7,545.8,568.4
XS GIS Cut Line= 3
     1951533.083       158529.28     1951818.835      158058.081
     1952489.727      157598.439
#Sta/Elev= 30
       0  2408.4   167.3 2398.28   226.3 2396.87   305.1    2393   403.5 2386.24
     433 2382.73   472.4 2375.29     492 2365.59   521.6 2355.74   551.1  2343.3
   580.8 2328.44   600.7 2320.24   610.6 2314.02   620.5 2310.61   660.2 2300.43
   719.7 2296.83   745.2 2297.05   765.2 2297.39   868.4 2297.99   957.7 2308.59
   977.5  2313.9   997.4 2321.48  1017.2 2332.17  1096.5 2364.57  1106.5 2370.86
  1116.4 2375.13  1195.7 2402.51  1205.6 2408.12  1235.4 2411.69  1364.3 2414.18
#Mann= 3 , 0 , 0
       0      .1       0   745.2    .045       0   765.2      .1       0
Bank Sta=745.2,765.2
XS Rating Curve= 0 ,0
Exp/Cntr=0.3,0.1

Type RM Length L Ch R = 1 ,28478.3 ,323.7,314,304.2
XS GIS Cut Line= 3
     1951558.625      158606.795     1951777.049      158343.617
     1952386.001      158498.319
#Sta/Elev= 30
       0 2407.35    78.2 2402.96    97.7 2399.83     215 2403.08   234.5 2400.21
   283.4 2386.83     342 2372.69     352 2365.95     362 2361.23   401.8 2345.61
   421.8 2336.42   441.7  2318.9   461.7 2307.19   481.6 2297.28   521.5 2283.08
   551.4 2282.41   554.4 2282.43   574.4 2282.69   601.3 2283.44   641.2 2288.64
   671.1 2295.72   681.1 2298.96     701 2311.27   760.9 2332.51   780.8 2343.01
   850.6 2366.23   860.6 2372.46   880.6 2375.75   930.4 2378.91   970.3 2384.52
#Mann= 3 , 0 , 0
       0      .1       0   554.4    .045       0   574.4      .1       0
Bank Sta=554.4,574.4
XS Rating Curve= 0 ,0
Exp/Cntr=0.3,0.1

Type RM Length L Ch R = 1 ,28164.4 ,368.6,369.9,371.3
XS GIS Cut Line= 2
     1951569.471      158760.915     1952380.783      158632.247
#Sta/Elev= 30
       0 2414.55    49.5 2413.98    89.1 2404.16   128.7  2392.5   138.6 2386.96
   178.2 2370.62   207.8 2356.26   227.6 2337.37     287  2299.7   296.9 2290.56
   306.8  2279.5   316.7 2274.36   326.6 2271.16   362.9 2268.68   382.9 2268.54
     386 2268.53   405.8 2269.91   465.2 2281.15   475.1 2284.94   524.5 2295.56
   544.3 2302.17   554.2 2309.03   564.1 2313.77   623.5 2332.88   643.3 2341.39
   702.7 2356.72   722.5 2365.54   791.8 2383.37   811.6 2389.62   821.4 2390.33
#Mann= 3 , 0 , 0
       0      .1       0   362.9    .045       0   382.9      .1       0
Bank Sta=362.9,382.9
XS Rating Curve= 0 ,0
Exp/Cntr=0.3,0.1

Type RM Length L Ch R = 1 ,27794.4 ,439.5,411.8,387.9
XS GIS Cut Line= 3
     1951628.666      159118.236      1952025.31        159061.4
     1952424.253      158833.612
#Sta/Elev= 30
       0  2413.1      88 2413.45   146.6 2407.88   195.5 2401.22   205.2 2397.72
     215 2389.97   224.8 2379.53   234.6 2367.94   244.3 2352.01   273.6 2329.32
   322.5  2295.6   332.3 2283.69   347.6 2273.35   351.8 2271.09   361.6  2268.5
   367.6 2268.14   400.7 2267.88   410.7 2269.19   440.6 2277.21   490.6 2292.25
   510.6 2301.55   580.5 2324.86   590.4 2328.96   600.4 2336.51   640.4 2351.16
   670.3 2357.01   700.3 2366.97   710.3  2369.1   810.2 2380.85   860.1 2389.43
#Mann= 3 , 0 , 0
       0      .1       0   347.6    .045       0   367.6      .1       0
Bank Sta=347.6,367.6
XS Rating Curve= 0 ,0
Exp/Cntr=0.3,0.1

Type RM Length L Ch R = 1 ,27382.6 ,410.1,399.9,386.8
XS GIS Cut Line= 3
     1952079.672      159728.684     1952221.996      159366.704
     1952485.923      158911.798
#Sta/Elev= 30
       0 2379.36    99.7 2378.74   109.7 2374.72   119.7  2366.8   129.6 2361.52
   139.6 2348.46   149.6 2339.53   189.5 2320.77   209.4 2308.68   229.4 2301.29
   259.3 2285.56   289.2 2274.15   309.2 2268.83   349.1  2267.9     379 2267.92
     399 2268.58   438.6 2274.62   488.2 2288.52   527.9 2303.63   537.8 2306.15
   547.7 2306.03   627.1 2325.41     637 2327.18   686.6 2329.88   756.1 2343.84
     766  2342.5   815.6 2348.96   875.2 2353.02     895 2358.29   914.9 2365.35
#Mann= 3 , 0 , 0
       0      .1       0     379    .045       0     399      .1       0
Bank Sta=379,399
XS Rating Curve= 0 ,0
Exp/Cntr=0.3,0.1

Type RM Length L Ch R = 1 ,26982.6 ,531.8,515.3,497.9
XS GIS Cut Line= 3
     1952591.886      159906.943     1952579.474      159527.788
     1952583.041      158947.798
#Sta/Elev= 30
       0 2386.35    49.9  2387.6   109.8 2387.44   149.8 2386.05   159.7 2384.96
   169.7 2381.55   189.7 2371.27   199.7 2369.92   219.6 2358.19   259.6  2336.5
   269.5 2329.45   289.5 2312.02   299.5 2309.95   329.4 2278.21   339.4 2269.24
   349.4 2264.47   359.4 2263.73   369.4 2263.83   389.4 2263.84   438.3 2264.49
   477.7 2269.18     635  2275.6   684.1  2280.1   752.9 2290.12   772.6 2291.93
   841.4 2305.35     861 2307.55   910.2 2318.72   949.5 2333.77   959.4 2334.59
#Mann= 3 , 0 , 0
       0      .1       0   369.4    .045       0   389.4      .1       0
Bank Sta=369.4,389.4
XS Rating Curve= 0 ,0
Exp/Cntr=0.3,0.1

Type RM Length L Ch R = 1 ,26467.2 ,471.6,476.3,480.9
XS GIS Cut Line= 3
     1953324.067      159617.282     1952720.669      159053.932
     1952679.279      158918.197
#Sta/Elev= 30
       0 2401.38   149.2 2401.72   228.8 2396.64   238.7 2395.08   248.6 2390.88
   258.6  2385.3   278.5 2376.96   308.3 2352.49   348.1 2310.91   387.9 2274.95
   397.8 2262.18   407.8  2253.3   417.7  2251.4   427.7  2251.2   465.7  2251.2
   485.7 2251.41   497.3 2252.08   537.1 2257.52   576.9 2261.01   646.5 2262.74
   745.9 2266.81   765.8 2270.75   815.6 2283.37     835 2286.04   853.9 2290.29
   901.2 2301.63   920.1 2307.64     939 2311.31     958 2318.37   967.4 2324.38
#Mann= 3 , 0 , 0
       0      .1       0   465.7    .045       0   485.7      .1       0
Bank Sta=465.7,485.7
XS Rating Curve= 0 ,0
Exp/Cntr=0.3,0.1

Type RM Length L Ch R = 1 ,25991   ,336.1,343.6,351.1
XS GIS Cut Line= 2
     1953462.902      159320.923     1952950.281      158389.126
#Sta/Elev= 30
       0  2335.6    49.7 2336.05    99.4 2334.31     159 2327.97   188.8 2315.52
   208.7 2311.74   238.5 2299.93   298.2 2268.95   308.1 2268.61   337.9 2252.42
   377.7 2244.35   397.6 2243.32   417.1 2243.36   437.1 2243.47   516.8 2250.55
   705.7 2254.33   755.4 2262.31   785.2 2265.24     825 2273.31   844.8  2281.6
   854.8 2283.02   864.7 2287.91   884.6 2304.34   924.4 2345.85   954.2 2365.65
     974 2371.85   993.9 2384.33  1013.8  2393.6  1043.6 2401.77  1063.5 2404.51
#Mann= 3 , 0 , 0
       0      .1       0   417.1    .045       0   437.1      .1       0
Bank Sta=417.1,437.1
XS Rating Curve= 0 ,0
Exp/Cntr=0.3,0.1

Type RM Length L Ch R = 1 ,25647.3 ,257.7,264.7,271.7
XS GIS Cut Line= 2
     1953633.573      159192.296     1953454.892      158327.719
#Sta/Elev= 30
       0 2278.46    29.8 2272.94    49.6 2271.87     129 2262.05   148.8 2260.83
   228.2 2250.34   238.1 2250.24   277.8 2245.55   327.4 2241.99   414.8 2238.72
   434.8 2238.66   476.1 2239.31   525.7 2250.42   535.7 2251.27   575.3    2264
   595.2 2273.45   605.1 2273.51   624.9 2282.84   634.9 2283.25   654.7 2292.86
   664.6 2299.71   694.4 2324.92   724.1 2353.25     734  2356.6     744 2361.88
   773.7 2386.18   793.6 2399.01   803.5 2402.44   813.4 2403.74   882.8 2407.62
#Mann= 3 , 0 , 0
       0      .1       0   414.8    .045       0   434.8      .1       0
Bank Sta=414.8,434.8
XS Rating Curve= 0 ,0
Exp/Cntr=0.3,0.1

Type RM Length L Ch R = 1 ,25382.6 ,754.8,747.1,739.4
XS GIS Cut Line= 3
     1953780.578      159172.466     1953811.203      158764.113
     1953841.829      158355.759
#Sta/Elev= 30
       0 2272.82      10 2271.45      40 2269.34   109.9 2258.17   129.8 2256.66
   199.8 2247.05   319.6 2238.94   359.6 2235.45   389.5  2234.6   399.5  2234.6
   419.5 2234.62   439.5 2235.66   489.4 2246.13   509.4 2248.32   559.3 2261.23
   579.3 2264.03   589.3 2267.01   609.3 2270.19   619.2  2274.5   629.2 2280.73
   669.2 2310.93   689.2 2327.17   699.2 2332.17   709.1 2335.88   739.1 2361.16
   769.1 2382.25     779  2388.3     789 2391.57     799 2393.21     819 2401.54
#Mann= 3 , 0 , 0
       0      .1       0   399.5    .045       0   419.5      .1       0
Bank Sta=399.5,419.5
XS Rating Curve= 0 ,0
Exp/Cntr=0.3,0.1

Type RM Length L Ch R = 1 ,24635.6 ,573.2,595.4,617.6
XS GIS Cut Line= 3
     1954656.349      159174.078     1954504.414      158530.702
     1954490.815      158191.554
#Sta/Elev= 30
       0 2315.32    78.9 2313.12   138.1  2308.2     148 2306.03   157.9 2301.78
   187.5 2285.93   207.2 2278.12   226.9 2275.33   286.1 2258.73     296 2256.38
   315.7 2254.33   374.9 2241.58   404.5 2233.78   414.4 2233.48   434.1 2228.91
   477.7 2227.42   483.5 2227.38   497.7  2227.6   621.6  2236.1     691 2242.62
   820.8 2248.44   850.8 2258.14   870.7 2266.61   890.7 2276.82   900.7 2277.74
   930.6 2293.28   950.6 2301.38   980.5 2311.32   990.5 2313.83  1000.5 2314.32
#Mann= 3 , 0 , 0
       0      .1       0   477.7    .045       0   497.7      .1       0
Bank Sta=477.7,497.7
XS Rating Curve= 0 ,0
Exp/Cntr=0.3,0.1

Type RM Length L Ch R = 1 ,24039.8 ,248.2,253.4,258.6
XS GIS Cut Line= 2
      1954791.77      159227.637     1955290.851      158574.785
#Sta/Elev= 30
       0 2308.35    69.3 2278.17    79.2 2274.15      99 2268.18   108.9 2262.84
   118.8 2259.16   148.5  2249.9   188.1 2239.38     198 2237.43   267.3 2230.28
     396 2222.78   429.6 2221.95   449.6 2221.88   465.3 2221.85   475.2 2222.36
   485.1 2224.95   564.3 2260.48   574.2 2262.21   584.2 2266.28   653.4 2300.92
   673.2 2307.64     693 2311.47   712.9 2317.87   762.4 2342.62   772.3 2349.05
   782.2 2356.83   792.1 2361.38     802 2368.54   811.9 2372.03   821.8 2377.35
#Mann= 3 , 0 , 0
       0      .1       0   429.6    .045       0   449.6      .1       0
Bank Sta=429.6,449.6
XS Rating Curve= 0 ,0
Exp/Cntr=0.3,0.1

Type RM Length L Ch R = 1 ,23786.4 ,910.9,935.6,960.4
XS GIS Cut Line= 3
     1954926.009      159320.923     1955366.852      158941.722
     1956226.252      158818.981
#Sta/Elev= 30
       0 2305.25    39.4 2293.39      69 2278.72   108.4 2265.49   128.1  2254.1
   246.4 2225.75   335.1 2216.06   424.3 2218.72   444.3 2218.71   463.2 2220.13
   492.8 2233.02   551.9 2262.58   571.6 2275.98   581.5 2285.25   601.4 2294.97
   631.4 2302.93   661.3 2306.97   711.2 2305.08     791 2297.81     831 2281.04
   890.8 2265.24   930.7 2258.94  1010.6 2270.94  1060.5 2287.34  1110.4 2296.93
  1210.1 2309.57    1290 2307.12  1309.9 2302.82  1389.7 2295.42  1449.6 2287.14
#Mann= 3 , 0 , 0
       0      .1       0   424.3    .045       0   444.3      .1       0
Bank Sta=424.3,444.3
XS Rating Curve= 0 ,0
Exp/Cntr=0.3,0.1

Type RM Length L Ch R = 1 ,22849.6 ,337.4,330.6,323.8
XS GIS Cut Line= 3
     1954947.368      159579.903     1955734.546      159731.716
     1956421.155      159243.495
#Sta/Elev= 30
       0 2301.91   108.9 2266.07   148.5 2249.73   168.2 2237.58   207.8 2223.91
   247.4 2213.09   297.8  2207.7   317.8 2206.22     386 2205.47   475.1 2211.39
   564.2 2228.26   643.3 2266.04   653.2 2279.71   682.9 2301.07   702.7 2307.53
   762.1 2314.49   781.9 2320.54   930.5 2397.46   960.3 2392.17   980.1 2394.26
  1059.4 2378.56    1099 2361.89  1128.8 2342.78  1148.6 2335.74  1198.2 2309.15
  1237.8 2294.08  1257.6 2290.99    1327 2288.81  1465.8 2305.03  1644.2 2311.34
#Mann= 3 , 0 , 0
       0      .1       0   297.8    .045       0   317.8      .1       0
Bank Sta=297.8,317.8
XS Rating Curve= 0 ,0
Exp/Cntr=0.3,0.1

Type RM Length L Ch R = 1 ,22518.5 ,359.9,355.6,351.6
XS GIS Cut Line= 2
     1954977.204      159967.639     1955863.145      159900.292
#Sta/Elev= 30
       0 2263.86    39.9 2252.14    49.9 2246.99    59.9  2243.5   119.8 2226.62
   129.8 2221.99   149.8 2216.36   209.6 2203.38   219.6 2201.86   249.6 2199.35
   279.5 2198.15   339.4 2201.26   399.8 2203.09   419.8 2203.05   439.3 2203.31
   509.1 2234.85   519.1 2239.77   539.1 2255.11     599 2287.02     609 2294.69
     619 2300.06   688.8 2302.79   698.8 2304.74   708.8 2308.73   728.8 2318.48
   768.7 2339.62   788.7 2356.24   848.6  2391.3   868.5 2407.02   888.5 2416.78
#Mann= 3 , 0 , 0
       0      .1       0   399.8    .045       0   419.8      .1       0
Bank Sta=399.8,419.8
XS Rating Curve= 0 ,0
Exp/Cntr=0.3,0.1

Type RM Length L Ch R = 1 ,22163.2 ,406.1,411.3,416.2
XS GIS Cut Line= 3
     1954984.747      160399.564       1955496.3      160272.613
     1955895.113       160179.72
#Sta/Elev= 30
       0 2264.82    29.8  2263.2    39.8 2261.55   109.4 2242.19   119.3 2238.88
   129.3 2232.84   139.2 2230.49   208.8 2222.04   298.3 2214.99   318.2 2211.85
   348.1 2204.13     368  2201.7   518.3 2202.46   527.1 2202.45   538.3 2205.98
     587 2230.28     597 2234.44     627 2244.17   656.9 2256.88   696.9 2277.98
   706.8 2284.83   716.8 2293.91   736.8  2302.9   746.8 2306.42   756.8 2308.66
   786.8 2310.23   856.7 2309.79   866.6 2308.83   896.6 2317.57   936.6 2332.73
#Mann= 3 , 0 , 0
       0      .1       0   518.3    .045       0   538.3      .1       0
Bank Sta=518.3,538.3
XS Rating Curve= 0 ,0
Exp/Cntr=0.3,0.1

Type RM Length L Ch R = 1 ,21751.8 ,689.5,699.9,710.3
XS GIS Cut Line= 2
     1955006.106      160674.564     1956044.698      160639.855
#Sta/Elev= 30
       0 2317.56      30 2311.71    89.9  2303.7   109.9 2296.07   179.9 2274.62
   199.8 2266.98   249.8 2251.74   259.8 2248.24   279.8 2237.71   289.8  2234.3
   339.7 2221.09   359.7 2213.32   369.7  2210.6   429.7 2198.52   449.6 2197.43
   487.6 2197.35   507.6 2196.86   549.6 2195.12   579.5 2195.85   609.5 2201.32
   659.5 2207.49   679.5 2212.38   739.4 2222.62   759.4 2227.16   819.4 2235.46
   839.3 2239.84   929.3 2254.01   989.2 2261.23  1009.2 2265.77  1039.2 2270.54
#Mann= 3 , 0 , 0
       0      .1       0   487.6    .045       0   507.6      .1       0
Bank Sta=487.6,507.6
XS Rating Curve= 0 ,0
Exp/Cntr=0.3,0.1

Type RM Length L Ch R = 1 ,21052.1 ,445.4,426.3,407.1
XS GIS Cut Line= 2
     1955160.465      161139.596     1955944.661      161465.686
#Sta/Elev= 30
       0 2330.18      30 2325.69      60 2312.26   109.9 2287.54   119.9 2282.33
   129.9  2274.8   199.8 2248.11   209.8 2242.23   219.8 2234.83   229.8 2228.76
   279.8 2211.52   289.8 2204.76   319.7 2194.45   339.7 2188.41   349.7 2186.43
   369.7 2185.72   431.6 2186.36   451.6 2186.35   459.6 2186.36   469.6 2187.61
   519.6 2201.65   559.5 2211.22   649.5  2218.4   679.4 2219.81   699.4 2222.34
   739.4 2230.44   799.3 2248.23   819.3 2253.33   829.3 2256.86   849.3 2260.62
#Mann= 3 , 0 , 0
       0      .1       0   431.6    .045       0   451.6      .1       0
Bank Sta=431.6,451.6
XS Rating Curve= 0 ,0
Exp/Cntr=0.3,0.1

Type RM Length L Ch R = 1 ,20625.3 ,332.5,327.1,322.3
XS GIS Cut Line= 3
      1954883.29      161857.331      1955713.63      161547.622
      1955996.64      161531.603
#Sta/Elev= 30
       0 2249.64    59.8 2241.22    69.7 2238.67   149.4 2228.66   169.3 2224.89
     239 2217.55   248.9 2215.33   258.9 2213.84   328.6 2206.04   338.6 2204.17
   408.3  2197.4   428.2  2194.6   497.9 2188.77   517.8 2185.49   537.7 2183.98
   557.9 2183.42   567.6  2183.4   577.9  2183.4   667.2 2183.61     707 2185.08
   746.8 2188.83   766.7 2191.73   866.3 2200.58   905.8 2203.62   974.2 2210.56
   993.7 2213.31  1013.3 2216.87  1101.3 2248.67  1150.1  2255.4  1169.7 2257.17
#Mann= 3 , 0 , 0
       0      .1       0   557.9    .045       0   577.9      .1       0
Bank Sta=557.9,577.9
XS Rating Curve= 0 ,0
Exp/Cntr=0.3,0.1

Type RM Length L Ch R = 1 ,20298   ,375.3,364.2,352.5
XS GIS Cut Line= 3
     1955221.934      162171.175     1955565.838      161949.209
     1955916.677      161736.254
#Sta/Elev= 30
       0 2301.52    49.9  2281.1    59.9 2275.92    69.9  2269.5    89.8 2260.14
   109.8 2251.99   129.8 2244.59   149.8 2241.86   159.7 2238.53   179.7 2228.92
   239.6 2209.15   259.6 2201.64   289.5 2191.98   299.5  2188.9   319.5 2186.19
   349.4 2178.86   359.4 2177.44   399.3 2176.89   419.3 2176.89   448.4 2176.04
   477.7 2176.02   536.4 2176.41   585.2 2178.86   634.1 2182.51   653.6 2185.64
     722 2194.85   731.8 2196.86   741.6  2199.7   800.2 2208.55   819.7 2212.34
#Mann= 3 , 0 , 0
       0      .1       0   399.3    .045       0   419.3      .1       0
Bank Sta=399.3,419.3
XS Rating Curve= 0 ,0
Exp/Cntr=0.3,0.1

Type RM Length L Ch R = 1 ,19933.9 ,613.5,625.7,638
XS GIS Cut Line= 3
     1955556.106      162578.205     1955700.281      162383.302
     1956028.679      161835.972
#Sta/Elev= 30
       0 2344.16    19.4 2340.81    38.8 2334.91    67.9 2322.22    87.3  2311.3
   116.4 2298.77   126.1 2295.66   135.8 2294.32   203.6 2263.68   232.7 2247.22
   242.4 2245.06   252.4 2241.25   292.3 2220.24   352.1 2193.82   362.1 2192.72
   382.1 2183.33     412    2172     422 2170.48   434.3 2170.44   454.3 2170.48
   541.6 2167.04   601.5 2169.48   651.3 2182.06   671.3 2185.62   691.2 2186.65
     761 2199.47     791 2206.02   810.9 2208.62   830.9 2214.15   880.7 2231.14
#Mann= 3 , 0 , 0
       0      .1       0   434.3    .045       0   454.3      .1       0
Bank Sta=434.3,454.3
XS Rating Curve= 0 ,0
Exp/Cntr=0.3,0.1

Type RM Length L Ch R = 1 ,19307.5 ,210.1,209.5,207.8
XS GIS Cut Line= 2
     1955953.265      162688.968     1956685.475      162260.486
#Sta/Elev= 30
       0 2264.15    39.9 2252.43    59.9 2249.31    79.8 2242.51   149.7 2225.34
   169.7 2222.01   179.6 2218.04   209.6  2210.3   239.5  2204.5   259.5 2199.48
   279.5 2192.34   349.3 2173.26   369.3 2165.85   376.8 2164.04   396.8 2161.61
   419.2 2161.43   439.2 2162.62   449.1  2166.6   459.1 2174.76   548.9 2223.66
   558.9 2232.16   568.9 2238.66   608.8 2253.51   618.8 2256.29   658.7 2263.95
   708.6  2262.8   738.6 2260.06   768.5 2259.72   788.5 2261.11   848.4 2259.14
#Mann= 3 , 0 , 0
       0      .1       0   376.8    .045       0   396.8      .1       0
Bank Sta=376.8,396.8
XS Rating Curve= 0 ,0
Exp/Cntr=0.3,0.1

Type RM Length L Ch R = 1 ,19098   ,387.2,400.6,418
XS GIS Cut Line= 3
     1956051.589       162883.22     1956406.576      162663.538
     1956743.476      162433.234
#Sta/Elev= 30
       0  2274.5    19.9 2271.19    39.8  2265.1    59.6 2261.86    69.6 2257.17
   149.1 2229.92     159 2224.42     169 2220.62   238.6 2198.15   258.4 2187.92
   268.4    2185   298.2 2177.33     328 2171.13   367.8 2164.08   407.5  2159.1
   427.4 2158.68   427.5 2158.68   447.3 2159.82   457.3 2166.25   487.1 2190.24
   536.9  2226.7   556.8 2248.08   566.8 2255.49   586.7 2263.69   656.4 2284.63
   686.2 2292.77   696.2 2294.48     726 2293.77   755.9 2296.53   825.6 2295.08
#Mann= 3 , 0 , 0
       0      .1       0   407.5    .045       0   427.5      .1       0
Bank Sta=407.5,427.5
XS Rating Curve= 0 ,0
Exp/Cntr=0.3,0.1

Type RM Length L Ch R = 1 ,18698   ,367.1,359.7,349.4
XS GIS Cut Line= 3
     1956085.839      162990.201     1956543.886      163024.647
     1956944.339       163084.74
#Sta/Elev= 30
       0 2268.49      10 2267.44      30 2257.78    89.9 2237.77    99.9 2232.28
   109.8 2228.21   129.8 2224.47   149.8 2222.21   219.7 2218.76   259.6 2211.89
   339.5 2187.77   359.5 2178.18   389.4 2169.12   429.4 2158.25   439.4 2156.68
   449.3 2156.63   469.3 2156.82   479.1 2157.72   498.8 2162.03   518.6 2169.74
   528.5 2171.55   587.7 2177.96   607.5 2182.18   627.2 2183.97   676.6 2191.46
   686.5 2194.23   696.4 2195.64   755.6  2201.2   834.6 2211.52   864.3 2217.51
#Mann= 3 , 0 , 0
       0      .1       0   449.3    .045       0   469.3      .1       0
Bank Sta=449.3,469.3
XS Rating Curve= 0 ,0
Exp/Cntr=0.3,0.1

Type RM Length L Ch R = 1 ,18337.2 ,511,512.1,513.1
XS GIS Cut Line= 2
     1956190.121      163465.354     1957008.534      163176.263
#Sta/Elev= 30
       0 2344.58      20 2342.17    39.9 2340.83   109.7 2339.39   119.7 2338.39
   129.7 2335.13   139.7 2329.68   159.6 2316.92   169.6 2309.61   179.6 2296.21
   249.4 2247.78   269.4 2226.53   339.2 2177.41   349.2 2165.03   359.2 2158.35
   369.1 2153.57   379.1 2151.85   404.2 2151.62     409  2151.6   424.2 2152.17
   478.9 2160.71   518.8 2163.81   548.7 2167.36   618.6 2171.99   658.5 2172.72
   688.4 2175.56   718.3 2180.52   768.2 2190.65   788.2 2196.29     868 2212.93
#Mann= 3 , 0 , 0
       0      .1       0   404.2    .045       0   424.2      .1       0
Bank Sta=404.2,424.2
XS Rating Curve= 0 ,0
Exp/Cntr=0.3,0.1

Type RM Length L Ch R = 1 ,17825   ,324.7,327,327.9
XS GIS Cut Line= 2
     1956386.615      163916.033     1957208.776      163662.185
#Sta/Elev= 30
       0 2342.25    19.8 2330.11    39.6 2319.61    59.3 2303.99   108.8 2276.12
   138.5 2262.26   148.4 2254.32   217.6 2224.48   237.4 2212.16   306.6 2183.41
   316.5 2175.72   385.7 2148.96   395.6 2147.27   404.8 2146.94   405.5 2146.92
   424.8 2146.98     455 2148.63   464.8 2150.79   474.7 2154.21   484.6 2158.88
   563.8 2172.37   583.5 2177.74   652.8 2191.67   662.6    2196   731.9 2213.94
   751.7 2220.99   791.2  2227.4   820.9 2234.62   830.8 2238.59   860.5  2245.3
#Mann= 3 , 0 , 0
       0      .1       0   404.8    .045       0   424.8      .1       0
Bank Sta=404.8,424.8
XS Rating Curve= 0 ,0
Exp/Cntr=0.3,0.1

Type RM Length L Ch R = 1 ,17498   ,511.2,495.8,481.8
XS GIS Cut Line= 3
     1956462.606      164195.188     1956863.932      164110.083
     1957259.129      164003.308
#Sta/Elev= 30
       0 2324.82    39.1  2308.9    58.6 2299.76    68.4 2290.95   136.8 2256.18
   146.5  2247.4   156.3  2240.5   214.9 2209.77   224.7 2203.39   234.4 2195.49
   302.8 2166.63   312.6 2159.74   332.1 2152.52   361.4 2145.08   390.7 2143.35
   400.3 2143.45   420.3 2144.75   470.2 2150.52   480.1  2153.5   490.1 2158.59
     560 2180.13     570 2186.06     580 2189.34     600 2194.73   639.9 2203.16
   659.9 2209.51   719.8 2222.35   739.7 2228.06   779.7 2231.37   819.6 2239.84
#Mann= 3 , 0 , 0
       0      .1       0   400.3    .045       0   420.3      .1       0
Bank Sta=400.3,420.3
XS Rating Curve= 0 ,0
Exp/Cntr=0.3,0.1

Type RM Length L Ch R = 1 ,17002.1 ,305.4,330.8,356.3
XS GIS Cut Line= 4
     1956469.213      164449.807     1956911.612      164689.349
     1957233.233      164343.408     1958404.893      164198.836
#Sta/Elev= 30
       0 2282.75    39.5 2272.47      69 2274.89     148 2263.09   236.8  2254.1
   276.2 2256.31     434 2230.72   463.6 2229.75   503.1 2223.62   522.8 2224.41
   552.3 2207.11     631 2146.73   640.9  2141.4   660.5  2139.2   669.4  2139.2
   689.4 2139.24   837.7 2152.18   926.2 2166.42  1005.2 2187.42  1094.5 2222.72
  1223.4 2254.55  1253.2 2265.83  1352.4 2289.21  1461.6 2303.64  1550.8 2302.35
    1660 2293.44  1848.4 2268.02  1997.3 2257.11  2076.6  2246.7    2156 2226.92
#Mann= 3 , 0 , 0
       0      .1       0   669.4    .045       0   689.4      .1       0
Bank Sta=669.4,689.4
XS Rating Curve= 0 ,0
Exp/Cntr=0.3,0.1

Type RM Length L Ch R = 1 ,16671.2 ,354.6,389.1,423.6
XS GIS Cut Line= 4
      1956557.32      164556.603     1956949.796      164807.574
     1957579.987      164924.541      1958482.32      164663.399
#Sta/Elev= 30
       0 2228.35    59.5 2227.55   188.3 2218.28   218.1  2219.9   297.4 2211.18
   376.6 2195.94   465.9 2186.03   544.7 2182.59   603.9 2166.11   623.6 2146.86
   646.1 2136.96   663.1 2135.78   666.1 2135.79   692.7 2136.07   751.8 2147.95
   860.3  2186.4   909.6 2207.45   939.2 2214.28    1097 2206.62  1206.7 2213.59
  1306.7 2206.34  1376.6 2206.71  1466.6 2212.51  1566.5 2225.58  1636.4 2227.65
  1736.4 2243.79  1896.3 2251.46  1976.2 2260.82  2016.2 2269.54  2046.2 2268.65
#Mann= 3 , 0 , 0
       0      .1       0   646.1    .045       0   666.1      .1       0
Bank Sta=646.1,666.1
XS Rating Curve= 0 ,0
Exp/Cntr=0.3,0.1

Type RM Length L Ch R = 1 ,16281.9 ,500.3,498.1,495.9
XS GIS Cut Line= 3
     1956437.174      164516.554      1956832.32      164764.855
     1956840.374      165381.946
#Sta/Elev= 30
       0 2250.19    19.9 2236.66    49.6 2222.53    99.3  2208.7   119.2 2213.99
   188.7 2203.72   208.5 2205.45   268.1 2202.41   297.9 2209.24   357.5 2207.57
   407.1 2203.11   476.6 2192.83   546.3 2164.46   566.2 2160.92   635.9 2141.34
   685.7  2134.9   722.7    2134   725.5 2133.98   742.7 2136.95   765.3 2148.56
   785.2 2154.06   854.9 2200.54   874.8 2207.51   894.7  2219.7   904.7 2221.93
   934.5 2239.38   944.5 2239.43   984.3 2231.11    1044 2214.75  1083.8 2215.31
#Mann= 3 , 0 , 0
       0      .1       0   722.7    .045       0   742.7      .1       0
Bank Sta=722.7,742.7
XS Rating Curve= 0 ,0
Exp/Cntr=0.3,0.1

Type RM Length L Ch R = 1 ,15783.8 ,732.7,724.3,715.9
XS GIS Cut Line= 2
     1956349.371      164427.335     1956407.805      165322.865
#Sta/Elev= 30
       0 2296.03    39.9 2282.64    59.8 2279.06    89.7 2266.51   109.7 2256.05
   139.6 2237.21   149.6 2235.01   159.5 2230.05   189.5  2209.3   209.4 2197.34
   229.3 2187.54   249.3 2181.99   289.2  2159.6   319.1 2146.38   329.1 2142.72
     349 2139.51     369 2133.99   398.9  2131.5   414.9 2131.61   434.9 2132.08
   508.6 2145.52   538.5 2148.07   588.3 2164.28   608.3 2169.34   678.1 2173.82
   727.9 2181.45   777.8 2186.23   837.6 2197.49   857.6 2199.56   897.4 2208.48
#Mann= 3 , 0 , 0
       0      .1       0   414.9    .045       0   434.9      .1       0
Bank Sta=414.9,434.9
XS Rating Curve= 0 ,0
Exp/Cntr=0.3,0.1

Type RM Length L Ch R = 1 ,15058.9 ,354.7,360.9,366.8
XS GIS Cut Line= 3
     1955710.961      164700.778     1955796.397      164860.972
     1956109.801      165566.411
#Sta/Elev= 30
       0 2278.13    47.8 2265.53   124.2 2248.66   143.3 2241.59   201.4 2229.53
     231 2221.88   270.6 2206.29   280.5 2204.77   290.4 2200.63   310.2 2187.44
   320.1 2182.88   369.6 2164.45   409.2 2152.52   419.1 2151.88   468.6 2139.18
   508.1    2127   526.5 2125.56   537.8 2125.04   546.5 2125.04   577.4 2125.82
     617  2134.6   636.8  2137.2   686.3 2150.68   706.1  2158.4   725.9 2168.02
   745.6 2172.55   824.8 2203.65   834.7 2204.68     904 2230.22   953.5 2245.98
#Mann= 3 , 0 , 0
       0      .1       0   526.5    .045       0   546.5      .1       0
Bank Sta=526.5,546.5
XS Rating Curve= 0 ,0
Exp/Cntr=0.3,0.1

Type RM Length L Ch R = 1 ,14698   ,463.5,459,454.8
XS GIS Cut Line= 3
      1955529.45      164872.961     1955599.922       165276.08
     1955673.414       165680.23
#Sta/Elev= 30
       0 2351.75    59.9 2304.64    69.9 2299.04    79.8 2297.94    89.8 2294.43
   149.7 2258.09   189.6 2232.15   199.6  2231.7   289.5 2176.56   299.4 2175.47
   319.4 2164.33   329.4 2162.98   339.4 2158.07   389.3 2126.95   399.2 2124.87
   419.2  2120.5   428.8 2120.31   448.4 2120.67   467.9 2123.84   487.5 2129.68
     507 2132.63   585.3 2152.42   595.1 2152.72     644 2163.97   683.1  2174.7
   702.6 2178.01   771.1 2202.87   780.9 2205.86   790.7 2206.86     820 2217.52
#Mann= 3 , 0 , 0
       0      .1       0   399.2    .045       0   419.2      .1       0
Bank Sta=399.2,419.2
XS Rating Curve= 0 ,0
Exp/Cntr=0.3,0.1

Type RM Length L Ch R = 1 ,14238.9 ,346,340.8,334.5
XS GIS Cut Line= 3
     1955023.792      165035.748     1955164.546      165420.298
     1955305.299      165804.848
#Sta/Elev= 30
       0 2288.84      20 2278.78      40 2274.09    89.9 2248.99   129.8 2225.87
   139.8 2224.55   159.8 2214.96   179.8 2209.73   209.7 2192.34   239.7  2171.3
   249.7 2170.01   279.7 2148.55   289.6 2142.15   299.6 2137.33   329.6 2126.03
   349.6 2123.14   379.5 2115.78   389.5  2115.4     400 2115.42     420 2116.38
   439.5 2121.51   449.4 2122.14   469.4 2126.45   499.4 2129.39   529.4 2133.72
   569.3  2135.5   679.2 2145.16   739.1 2155.63   749.1 2155.92     819 2167.59
#Mann= 3 , 0 , 0
       0      .1       0     400    .045       0     420      .1       0
Bank Sta=400,420
XS Rating Curve= 0 ,0
Exp/Cntr=0.3,0.1

Type RM Length L Ch R = 1 ,13898   ,402.7,400,398.3
XS GIS Cut Line= 3
     1954631.921      165196.038     1954847.718      165543.068
     1955081.248      165883.706
#Sta/Elev= 30
       0 2303.61      10 2299.66    49.8 2269.57    69.8 2256.24    79.7 2252.61
    89.7  2250.3   119.6 2221.76   129.6 2213.75   139.5 2207.59   179.4 2185.92
   189.4 2184.61   199.3 2180.82   229.2 2165.83   259.2 2152.73   279.1 2143.16
     299 2136.13     309 2135.31   398.7 2112.74   418.7 2111.64   428.3 2111.62
     448 2112.01   457.8 2113.58   487.3 2120.83   497.2 2121.99   546.3 2125.49
   605.3 2131.43   654.5 2134.96   723.3 2141.87   772.5 2145.53   821.7 2154.35
#Mann= 3 , 0 , 0
       0      .1       0   398.7    .045       0   418.7      .1       0
Bank Sta=398.7,418.7
XS Rating Curve= 0 ,0
Exp/Cntr=0.3,0.1

Type RM Length L Ch R = 1 ,13498   ,400.9,400,401.6
XS GIS Cut Line= 3
     1954320.695      165505.846     1954573.001      165828.523
     1954825.548       166150.84
#Sta/Elev= 30
       0 2223.69      30 2207.64      50 2198.79    69.9 2188.51   109.9 2173.39
   149.9    2160   159.8 2157.44   169.8 2156.34   189.8 2150.02   249.8 2135.71
   279.7 2130.02   299.7    2128   309.7 2125.76   369.6 2108.11   389.6 2105.62
   399.6 2105.63   419.6 2105.64   439.6  2108.2   479.5 2120.58   539.4 2130.02
   589.4  2143.7   599.4  2147.1   619.3 2157.49   639.3 2165.86   649.3 2168.08
   719.2 2191.82   749.2 2205.18   759.2 2208.67   779.1 2213.59   819.1 2226.32
#Mann= 3 , 0 , 0
       0      .1       0   399.6    .045       0   419.6      .1       0
Bank Sta=399.6,419.6
XS Rating Curve= 0 ,0
Exp/Cntr=0.3,0.1

Type RM Length L Ch R = 1 ,13098   ,402.6,400,396.1
XS GIS Cut Line= 3
      1953964.19      165715.548     1954227.691      166028.439
     1954460.442      166368.363
#Sta/Elev= 30
       0 2339.47    29.9 2340.55    39.9 2337.84    49.9 2329.73    69.8 2308.48
    79.8 2297.22    89.8 2283.79    99.8 2267.88   109.8 2256.74   129.7 2237.63
   139.7 2231.04   149.7 2227.57   229.5 2169.39   259.4 2154.22   269.4 2150.34
   279.4 2148.81   319.3 2130.34   379.1 2097.07   389.1 2094.92   399.1 2094.62
   418.9 2094.52   419.1 2094.53   428.7 2094.89   438.5 2097.48   467.9 2115.03
   497.3 2121.98   585.6 2134.03   742.6 2150.46   781.8 2158.03     821 2164.02
#Mann= 3 , 0 , 0
       0      .1       0   399.1    .045       0   419.1      .1       0
Bank Sta=399.1,419.1
XS Rating Curve= 0 ,0
Exp/Cntr=0.3,0.1

Type RM Length L Ch R = 1 ,12698   ,400.4,400,398.3
XS GIS Cut Line= 3
     1953626.085      166001.393     1953921.192      166285.149
     1954202.645      166583.403
#Sta/Elev= 30
       0 2329.64    89.9 2338.11    99.8 2334.42   109.8  2322.7   119.8 2307.28
   139.8 2270.85   159.8 2249.97   169.8 2234.52   179.7 2222.87   199.7 2201.25
   209.7 2188.56   219.7 2179.17   239.6 2163.59   269.6 2144.35   279.6 2139.06
   289.6 2134.85   299.6 2132.33   319.5 2122.84   339.5 2109.36   379.4 2086.98
   389.4 2083.54   399.4  2082.9   419.2 2082.88   419.4 2082.88   438.7 2084.51
   477.7 2102.36   497.3 2107.47   692.6 2129.05   760.9 2138.95   819.5 2149.31
#Mann= 3 , 0 , 0
       0      .1       0   399.4    .045       0   419.4      .1       0
Bank Sta=399.4,419.4
XS Rating Curve= 0 ,0
Exp/Cntr=0.3,0.1

Type RM Length L Ch R = 1 ,12298   ,397.8,399.9,399.5
XS GIS Cut Line= 3
     1953334.445      166284.978     1953634.524      166563.622
     1953934.604      166842.266
#Sta/Elev= 30
       0 2333.06      40 2336.37    49.9  2334.6    59.9 2326.55    79.9 2306.42
   139.8 2239.83   149.8 2233.14   179.8 2202.38   189.8 2193.66   209.7 2178.34
   229.7  2164.8   269.7 2140.09   279.7 2132.94   289.6 2128.82   299.6 2127.14
   349.6 2101.71   379.5 2084.39   389.5 2079.64   399.5 2079.55   409.5 2079.49
   419.5 2079.49   429.5 2079.86   439.5 2081.88   469.4 2093.62   499.4 2100.58
   559.3 2111.22   589.3 2114.93   649.2 2126.39   699.2 2132.93     819 2144.24
#Mann= 3 , 0 , 0
       0      .1       0   399.5    .045       0   419.5      .1       0
Bank Sta=399.5,419.5
XS Rating Curve= 0 ,0
Exp/Cntr=0.3,0.1

Type RM Length L Ch R = 1 ,11898   ,414.2,414.3,416.7
XS GIS Cut Line= 3
     1953126.016      166569.072     1953427.875      166899.331
     1953727.554      167168.489
#Sta/Elev= 30
       0 2246.03     9.9 2243.84    19.9 2238.74    79.5 2196.96   109.4 2173.14
   119.3 2164.15   139.2 2157.12   188.9 2124.48   228.7 2097.11   238.6 2091.79
   258.5 2086.38   308.2 2079.58   397.7  2071.1   437.4  2069.8   457.4    2071
   467.1 2073.78   476.9 2077.93   486.7  2084.5   506.4    2093   535.8 2102.04
   555.5  2105.7   575.1 2111.08   604.6 2120.64   673.4 2136.36     693 2139.44
   702.9 2142.77   791.3 2164.13   820.8 2172.21   840.4 2174.66   850.2  2176.9
#Mann= 3 , 0 , 0
       0      .1       0   437.4    .045       0   457.4      .1       0
Bank Sta=437.4,457.4
XS Rating Curve= 0 ,0
Exp/Cntr=0.3,0.1

Type RM Length L Ch R = 1 ,11483.6 ,226.6,237,246.5
XS GIS Cut Line= 2
     1952796.766      166786.235      1953348.06      167392.588
#Sta/Elev= 30
       0 2189.52      20 2181.14      70 2157.35      90 2152.95    99.9  2148.9
   109.9 2147.41   169.9  2121.1   219.9 2102.75   229.9 2100.14   239.9 2095.23
   309.8 2077.83   359.8 2068.75   399.5 2064.06   419.5 2063.68   429.7 2063.57
   449.7 2064.74   489.7  2070.2   539.7 2078.03   549.7 2080.02   559.7 2083.69
   599.6  2110.1   609.6 2119.15   629.6 2129.38   709.6 2199.66   719.6 2209.95
   729.6 2224.03   739.6 2230.68   749.6 2233.95   789.5 2261.28   819.5 2277.87
#Mann= 3 , 0 , 0
       0      .1       0   399.5    .045       0   419.5      .1       0
Bank Sta=399.5,419.5
XS Rating Curve= 0 ,0
Exp/Cntr=0.3,0.1

Type RM Length L Ch R = 1 ,11246.5 ,322.5,326.8,332.1
XS GIS Cut Line= 3
     1952763.204      166864.035     1952896.523      167258.067
     1953073.432      167626.115
#Sta/Elev= 30
       0 2168.87     9.9 2166.37    89.1 2132.16      99 2131.27   198.1 2101.97
     208 2101.09   267.4 2080.24   287.2 2075.02   356.6 2061.45   386.3 2060.25
   387.6 2060.27   407.6 2060.85   425.9 2065.23   455.8 2076.17   495.6 2103.47
   505.6 2103.82   575.3 2143.68   605.2 2163.31   615.2  2164.6   625.1 2169.95
     665 2199.25   684.9 2216.61   704.8 2236.58   714.8 2237.13   724.7 2246.26
   734.7 2261.17   744.6 2273.57   754.6 2279.58   794.4 2289.52   824.3 2293.05
#Mann= 3 , 0 , 0
       0      .1       0   387.6    .045       0   407.6      .1       0
Bank Sta=387.6,407.6
XS Rating Curve= 0 ,0
Exp/Cntr=0.3,0.1

Type RM Length L Ch R = 1 ,10919.6 ,609.2,611.7,614.1
XS GIS Cut Line= 2
     1952515.086       166855.39     1952648.581      167765.827
#Sta/Elev= 30
       0 2278.07    29.7  2272.7    49.5 2260.66      89 2230.06   108.8 2222.42
   168.2 2181.08   178.1  2172.6   197.9 2150.46   207.8 2147.76   227.6 2124.37
   237.5 2115.87   267.2 2098.93   286.9 2090.74   296.8 2090.55   356.2 2074.48
   405.7  2067.4   474.9 2053.58     496 2052.83   514.5 2052.71     516 2052.82
   534.3 2056.34     564 2072.78   583.8 2078.86   672.8 2135.57   682.7 2136.81
   761.9 2191.94   771.8 2192.35   831.1 2234.84     841 2239.78   920.2 2250.23
#Mann= 3 , 0 , 0
       0      .1       0     496    .045       0     516      .1       0
Bank Sta=496,516
XS Rating Curve= 0 ,0
Exp/Cntr=0.3,0.1

Type RM Length L Ch R = 1 ,10307.8 ,394.1,409.8,419.8
XS GIS Cut Line= 2
     1951970.386       166936.58     1952010.475      167749.807
#Sta/Elev= 30
       0 2177.48     9.9 2173.24    29.8 2169.07    59.6 2156.45    99.3 2142.89
   119.2 2140.28   198.6 2121.72   218.4 2119.19   258.2 2108.64   307.8 2091.26
   347.5  2066.9   377.3 2051.02   387.2 2047.34   402.8 2045.96     417  2045.8
   422.8 2045.82   436.9 2046.39   446.8 2048.47   476.6  2057.2   546.1 2061.14
     556 2063.08     566 2068.22   585.8 2081.61   595.8 2083.18   675.2 2139.42
   685.1 2140.32   714.9 2162.41   764.6 2202.26   774.5  2202.7   814.2 2232.82
#Mann= 3 , 0 , 0
       0      .1       0   402.8    .045       0   422.8      .1       0
Bank Sta=402.8,422.8
XS Rating Curve= 0 ,0
Exp/Cntr=0.3,0.1
